HEC-RAS study 2027_ras.prj: 2027

--- 2027_ras.g01 (geometry) --- (continued)

Type RM Length L Ch R = 1 ,32688.71,247.946600,247.946600,247.946600
XS GIS Cut Line= 6
605879.813047917733078.001943868 605015.13034296733307.901557595
604408.521008104733626.980651483604089.880480587733971.145991802
603817.190039426734716.223194525603135.633122414735078.462525085
#Sta/Elev= 30
7580.798177.6547 7821.11177.86647892.163172.00778057.789175.19358078.476167.7697
8234.328170.81348276.196175.47358530.074176.08018572.977171.46038752.114170.8458
8775.019165.66198859.931163.03299022.301164.31029193.167158.04379396.758159.5712
9425.969151.3304 9503.38151.66699581.326175.34689607.158174.17049663.194155.6011
9685.855153.249910100.55 152.83610110.78153.314910152.03169.749910215.59175.7702
10506.41173.246210731.79185.829510975.75185.862211195.29202.920811225.55213.4663
#Mann= 3 , 0 , 0
7580.798  0.0712       07580.798  0.0712       011225.55  0.0712       0
#XS Ineff= 2 , 0
       09585.622                       0
Bank Sta=7580.798,11225.55
Exp/Cntr=0.3,0.1

Type RM Length L Ch R = 1 ,32440.76,247.946600,247.946600,247.946600
XS GIS Cut Line= 6
605892.388055793 733022.08329181605041.323814332733226.926045194
604380.046954155733532.096171364603983.666884542 733879.27350086
603531.768886715734553.471571699602953.201436013 734881.51834701
#Sta/Elev= 30
7425.464178.58717872.488173.53917934.258  169.15 8068.41170.31558120.232174.6085
 8445.54175.20848606.963170.64998628.695165.49148966.919158.83069236.547156.9506
9286.282 162.1159311.483152.4579 9342.28150.83719397.692152.74729474.617175.3958
9498.351173.30829543.523153.98659554.872151.86079997.112150.834210145.87153.0712
10206.82171.260310479.64 178.07210568.13 176.71410628.44185.629110721.37187.2677
 10810.8209.111510919.04229.6111 10972.4242.035911014.36255.321711047.71253.9294
#Mann= 3 , 0 , 0
7425.464   0.044       07425.464   0.044       011047.71   0.044       0
#XS Ineff= 2 , 0
       09478.566                       0
Bank Sta=7425.464,11047.71
Exp/Cntr=0.3,0.1

Type RM Length L Ch R = 1 ,32192.82,247.946500,247.946500,247.946500
XS GIS Cut Line= 6
 605899.39639025732990.918570498605193.335839331 733143.38677609
604618.035763711733342.495730653604235.052266866733557.140421763
603323.486545384734233.065911412602608.393221825734530.660865888
#Sta/Elev= 30
7391.252178.6111 7517.93178.6205 7548.48174.81927619.764177.53967885.609169.2102
8029.542170.1469  8081.1174.21858414.906173.88278553.223 170.8638585.405166.0879
 9162.84156.16519279.295162.39289323.564150.51279348.973150.1771 9399.79153.1208
9464.859177.87799491.084173.86919549.427152.673710037.53149.093710264.91 149.634
10323.25153.614610390.03173.466910503.25 169.25110533.74173.709510625.29173.9224
10840.49187.993310882.62193.582610955.99210.246811008.06229.3728 11076.9263.7362
#Mann= 3 , 0 , 0
7391.252  0.0434       07391.252  0.0434       0 11076.9  0.0434       0
#XS Ineff= 2 , 0
       09474.865                       0
Bank Sta=7391.252,11076.9
Exp/Cntr=0.3,0.1

Type RM Length L Ch R = 1 ,31944.87,247.946600,247.946600,247.946600
XS GIS Cut Line= 6
 605908.20080063732951.767043478604874.708409131733184.682090655
604378.229072869733384.727258429603583.922026455733814.518682927
 602692.20018062734085.535117745602195.407658339  734182.4648422
#Sta/Elev= 30
7382.982178.64137620.205178.19437895.448169.52568234.705174.03198484.948171.7715
8665.278163.43219044.502160.75169061.496158.13479164.736156.09629303.944160.2518
9325.283156.78739339.008148.66919350.696148.22929432.512152.02119479.264171.7638
 9502.64177.62669525.903173.17769560.572  158.819595.241 151.4779966.426148.2114
   10553151.2982 10594.8153.353810657.16164.0472 10760.8163.428510813.48 169.558
10874.25170.673210884.51173.626610905.05185.856410915.32186.819411321.91201.5781
#Mann= 3 , 0 , 0
7382.982  0.0401       07382.982  0.0401       011321.91  0.0401       0
#XS Ineff= 2 , 0
       09509.926        10291.37       0
Bank Sta=7382.982,11321.91
Exp/Cntr=0.3,0.1

Type RM Length L Ch R = 1 ,31696.92,247.946600,247.946600,247.946600
XS GIS Cut Line= 6
605920.514667665732897.009634739604813.886008322 733120.50900209
604487.093104571733224.980345041603571.605765283733577.495950103
602462.367526323733788.223661616601699.425913721733863.311371744
#Sta/Elev= 30
7390.268178.68367659.473178.10937903.462168.8447 8529.03171.73758622.783169.4191
8738.162153.98269341.744158.47069428.842147.04339515.509149.02189568.948174.1087
9579.634174.32169611.692172.15159664.602154.96859820.932146.834810300.04150.2049
10340.83154.786210391.81173.8202 10432.6174.671210483.59166.030510554.97176.4275
10646.75154.0095 10839.9150.6228 10870.3153.921710910.83165.875411022.11165.7364
11314.42179.8605 11475.1198.592211595.44222.297911645.54 227.90411741.26211.0309
#Mann= 3 , 0 , 0
7390.268    0.04       07390.268    0.04       011741.26    0.04       0
#XS Ineff= 2 , 0
       0 9701.34        10198.32       0
Bank Sta=7390.268,11741.26
Exp/Cntr=0.3,0.1

Type RM Length L Ch R = 1 ,31448.98,247.946600,247.946600,247.946600
XS GIS Cut Line= 6
 605937.06042165732823.433835091604706.166111827733032.188347444
603699.461322516733296.846674278603037.451922297733421.636378109
602319.474933147733511.835255548601523.561968744733549.960443333
#Sta/Elev= 30
7379.378178.74037867.117168.05668506.824171.67088629.243 167.6368742.202152.1371
9342.375153.38999601.482142.65099663.399169.37129724.951175.38079847.763172.9095
9888.518145.724810122.33145.603410132.47150.818410142.61 173.72810162.89174.0805
 10264.3174.031310365.69152.318710497.09152.870110567.87182.551210588.06183.8249
10628.38183.464510698.95160.830610819.91176.180110930.48157.305211101.27157.6765
11201.57172.212911321.87170.759111622.19187.129411752.25208.4553 11863.7236.9872
#Mann= 3 , 0 , 0
7379.378    0.04       07379.378    0.04       0 11863.7    0.04       0
#XS Ineff= 2 , 0
       09758.652        10245.34       0
Bank Sta=7379.378,11863.7
Exp/Cntr=0.3,0.1

Type RM Length L Ch R = 1 ,31201.03,247.946600,247.946600,247.946600
XS GIS Cut Line= 6
 605953.93241085 732748.40732991603964.731713086733007.895050585
 603118.43428731733161.094618291602936.275880009733185.638160393
602197.227419078733233.698224172601356.965753883733234.343899906
#Sta/Elev= 30
7350.052178.96088326.976167.76868679.714159.09178740.183150.99739406.427152.7148
9689.921137.74879771.235151.59189924.253144.30079944.719129.18249985.651119.1763
10047.02 122.85110067.47140.923410229.98150.555910270.34141.710110461.78  154.18
 10552.2176.182310592.38178.669610612.47175.242810642.55157.966910792.87162.7898
10933.09154.275110993.14175.257111033.17178.291711163.25176.188711233.26164.1276
11453.29169.8359 11623.3205.6509 11793.3228.533311893.32 227.65811981.37209.9908
#Mann= 3 , 0 , 0
7350.052  0.0537       07350.052  0.0537       011981.37  0.0537       0
#XS Ineff= 2 , 0
       09787.622        10196.46       0
Bank Sta=7350.052,11981.37
Exp/Cntr=0.3,0.1

Type RM Length L Ch R = 1 ,30953.08,247.946600,247.946600,247.946600
XS GIS Cut Line= 6
605966.679191962732691.724835165 604903.98170197732799.525323182
 603552.94052577732852.576341927602951.945520639 732903.68947196
602216.673486143732895.764945492600252.414384186732802.726766437
#Sta/Elev= 30
7305.893178.35098202.581168.67028683.705159.03128723.764150.60419344.072152.7564
9754.401136.13169814.572145.67079864.715142.99899904.836 129.2819975.387120.5994
10066.13 126.41910116.39142.954110216.66139.796710286.72153.887910386.77156.6667
10436.78165.187910486.79165.865710506.79155.5589 10746.8154.734611066.92161.2827
11187.04 180.32111377.21180.396411467.29168.715111537.36177.818711587.42170.3428
12318.36177.829612338.38183.934612438.51180.995312939.05198.641213031.72208.4788
#Mann= 3 , 0 , 0
7305.893  0.0583       07305.893  0.0583       013031.72  0.0583       0
#XS Ineff= 2 , 0
       09749.978        10155.49       0
Bank Sta=7305.893,13031.72
Exp/Cntr=0.3,0.1

Type RM Length L Ch R = 1 ,30705.14,247.946600,247.946600,247.946600
XS GIS Cut Line= 6
605975.978496493732650.372608627604902.823034644732740.116884857
604137.386846066732727.220418304603438.510168761732664.843635455
601678.860253751732410.252431467  600198.8945494732303.690469265
#Sta/Elev= 30
7300.267177.97427603.075177.6172 7773.92168.41347914.378170.31688365.284160.4671
8685.352158.68368735.354150.19779045.592151.77419195.907 147.5799276.144156.0652
9316.263149.7513 9436.62148.83959526.902141.79179788.165140.72699838.574135.6628
9868.958142.6124  9929.9 125.1189981.355120.883210074.37124.570410125.35140.6404
10176.06138.479610216.56149.944810287.36154.177410670.89148.148311094.54152.3102
11134.85155.772611175.15167.640111215.46 173.26812421.23182.309313108.38199.7902
#Mann= 3 , 0 , 0
7300.267  0.0473       07300.267  0.0473       013108.38  0.0473       0
#XS Ineff= 2 , 0
       09759.101         10214.1       0
Bank Sta=7300.267,13108.38
Exp/Cntr=0.3,0.1

Type RM Length L Ch R = 1 ,30457.19,247.946500,247.946500,247.946500
XS GIS Cut Line= 6
605988.870122926732593.046014478605077.267775536732655.743316606
604460.328160286732627.062881216601837.495038599732075.717592731
601128.429862797 731988.22083357600158.813171595731929.958702967
#Sta/Elev= 30
 7328.33177.41857623.622178.29617804.171168.86887954.467171.00518424.678159.1824
8735.137159.12688785.376149.21329108.794150.85119611.689140.77259848.085141.0471
 9888.96137.08099929.643124.599410010.95121.157810082.16127.195310143.41144.3971
10235.77144.154510276.88149.4151 10453.5144.556211066.79148.112211158.45 149.745
11189.01164.3345 11260.3163.201511311.12169.045211463.29165.157411564.57166.4444
11584.79 171.63412570.81181.498813031.57181.275213091.61187.112113227.89187.7011
#Mann= 3 , 0 , 0
 7328.33  0.0523       0 7328.33  0.0523       013227.89  0.0523       0
#XS Ineff= 2 , 0
       09725.816        10272.67       0
Bank Sta=7328.33,13227.89
Exp/Cntr=0.3,0.1

Type RM Length L Ch R = 1 ,30209.25,1522.881100,1522.881100,1522.881100
XS GIS Cut Line= 6
605939.785761833732559.921089336605081.101253629732598.547520891
604477.344072998732540.859589666602164.577139974731715.883841261
601892.816451252731658.995914131600960.170907438731677.468872175
#Sta/Elev= 30
7395.691 176.9727571.079  178.297811.589 169.6998131.749169.29198662.847150.9535
  9039.6148.15059153.841150.6741  9483.7140.66779863.449138.81389896.023126.6837
9917.739123.41539961.742 124.3629994.767119.540810049.69123.479410093.59139.1846
10180.47141.682210493.54142.118110536.55145.802410653.94142.634711157.76143.0742
11240.39149.339211291.88158.9222 11527.3155.6447 11628.7158.098411648.71162.5397
11958.77161.222112008.78165.321612318.84 167.52812388.85174.186412533.71172.8491
#Mann= 3 , 0 , 0
7395.691  0.0504       07395.691  0.0504       012533.71  0.0504       0
#XS Ineff= 2 , 0
       0 9690.42        10200.68       0
Bank Sta=7395.691,12533.71
Exp/Cntr=0.3,0.1

Type RM Length L Ch R = 1 ,28686.36,148.643100,148.643100,148.643100
XS GIS Cut Line= 6
 605281.97921443731618.558292061604657.949096978731371.195002243
604460.616562307731128.104198635603825.720581084730676.241293117
601952.380966812 731175.79852356601034.684873432731360.784516826
#Sta/Elev= 30
8782.903154.24689349.774139.41179815.618133.72029844.037135.50739867.355131.5454
9893.133120.48019917.681119.46819936.339115.43159988.076121.854810040.42116.1138
10089.52130.657910114.07131.808210482.29132.120310543.66129.565910762.78130.6209
10907.68128.253911280.26130.768511601.09126.805311890.87127.581712149.61136.1306
12460.09137.481212501.38139.554712582.99151.9194 12674.8150.048312705.41153.7919
12980.84155.816413093.05158.916213154.26164.121113266.47163.352513430.01170.5305
#Mann= 3 , 0 , 0
8782.903  0.0518       08782.903  0.0518       013430.01  0.0518       0
#XS Ineff= 2 , 0
       09804.186        10140.74       0
Bank Sta=8782.903,13430.01
Exp/Cntr=0.3,0.1

Type RM Length L Ch R = 3 ,28594.04,,,
BEGIN DESCRIPTION:
END DESCRIPTION:
Bridge Culvert--1,0,-1,-1, 0
Deck Dist Width WeirC Skew NumUp NumDn MinLoCord MaxHiCord MaxSubmerge Is_Ogee
48.321550,52.000000,2.6,0, 60, 60, , , 0.95, 0, 0,0,,
 8879.62 8899.74 8931.80 8995.92 9017.29 9038.66 9049.35 9060.03 9070.72 9092.09
 9113.46 9145.52 9166.89 9188.27 9198.95 9221.29 9241.70 9348.51 9363.59 9412.53
 9444.54 9465.88 9487.22 9498.96 9528.31 9572.34 9610.03 9631.04 9673.24 9719.05
 9768.36 9787.77 9810.68 9824.87 9862.55 9869.63 9869.63 9872.2010086.6310086.63
10167.4610180.1710192.8710205.5810243.0610265.9010375.6110399.7110423.8110447.91
10472.0210484.0710508.1710532.2710568.4210592.5210604.5710616.6210628.6710632.77
  149.44  147.73  145.42  142.39  141.72  141.42  141.05  141.08  140.83  140.64
  140.18  139.68  139.54  139.31  139.09  138.94  138.65  137.77  137.87  137.61
  137.87  137.64  137.56  137.67  137.61  137.44  137.16  137.20  137.00  137.27
  137.98  138.00  138.24  138.27  137.90  137.06  137.06  136.75  136.52  136.52
  136.47  136.28  135.90  135.66  135.17  134.72  131.73  131.49  131.00  131.03
  130.61  130.60  130.37  129.88  129.73  129.19  129.03  129.13  129.01  129.06
 -850.56 -852.27 -854.58 -857.61 -858.28 -858.58 -858.95 -858.92 -859.17 -859.36
 -859.82 -860.32 -860.46 -860.69 -860.91 -861.06 -861.35 -862.23 -862.13 -862.39
 -862.13 -862.36 -862.44 -862.33 -862.39 -862.56 -862.84 -862.80 -863.00 -862.73
 -862.02 -862.00 -861.76 -861.73 -862.10 -862.94  133.06  132.75  132.52 -863.48
 -863.53 -863.72 -864.10 -864.34 -864.83 -865.28 -868.27 -868.51 -869.00 -868.97
 -869.39 -869.40 -869.63 -870.12 -870.27 -870.81 -870.97 -870.87 -870.99 -870.94
 8879.62 8899.74 8931.80 8995.92 9017.29 9038.66 9049.35 9060.03 9070.72 9092.09
 9113.46 9145.52 9166.89 9198.95 9221.29 9241.70 9348.51 9363.59 9412.53 9444.54
 9465.88 9487.22 9498.96 9528.31 9572.34 9610.03 9631.04 9673.24 9719.05 9768.36
 9787.77 9810.68 9824.87 9862.55 9872.20 9930.09 9930.0910147.0910147.0910167.46
10180.1710192.8710205.5810255.1110291.2610301.7410375.6110399.7110423.8110447.91
10472.0210484.0710508.1710532.2710568.4210592.5210604.5710616.6210628.6710632.77
  149.44  147.73  145.42  142.39  141.72  141.42  141.05  141.08  140.83  140.64
  140.18  139.68  139.54  139.09  138.94  138.65  137.77  137.87  137.61  137.87
  137.64  137.56  137.67  137.61  137.44  137.16  137.20  137.00  137.27  137.98
  138.00  138.24  138.27  137.90  136.75  136.69  136.69  136.45  136.45  136.47
  136.28  135.90  135.66  134.95  133.98  133.80  131.73  131.49  131.00  131.03
  130.61  130.60  130.37  129.88  129.73  129.19  129.03  129.13  129.01  129.06
 -850.56 -852.27 -854.58 -857.61 -858.28 -858.58 -858.95 -858.92 -859.17 -859.36
 -859.82 -860.32 -860.46 -860.91 -861.06 -861.35 -862.23 -862.13 -862.39 -862.13
 -862.36 -862.44 -862.33 -862.39 -862.56 -862.84 -862.80 -863.00 -862.73 -862.02
 -862.00 -861.76 -861.73 -862.10 -863.25 -863.31  132.69  132.45 -863.55 -863.53
 -863.72 -864.10 -864.34 -865.05 -866.02 -866.20 -868.27 -868.51 -869.00 -868.97
 -869.39 -869.40 -869.63 -870.12 -870.27 -870.81 -870.97 -870.87 -870.99 -870.94
Pier Skew, UpSta & Num, DnSta & Num=  ,9941.30, 2 ,10001.75, 2 , 0 , 0 , 0 ,,
    4.00    4.00
 -863.32  136.68
    4.00    4.00
 -863.39  136.61
Pier Skew, UpSta & Num, DnSta & Num=  ,10014.96, 2 ,10075.42, 2 , 0 , 0 , 0 ,,
    4.00    4.00
 -863.40  136.60
    4.00    4.00
 -863.47  136.53
BR Coef=-1 , 0 , 0 ,, 0 ,,,0.8,0,1,0,
WSPro=,,,, 1 ,,,, 0 ,,,, 0 ,,,,-1 ,-1 ,-1 , 0 , 0 , 0 , 0 , 0
BC Design=,, 0 ,, 0 ,,,,,,

Type RM Length L Ch R = 1 ,28537.72,855.736000,855.736000,855.736000
XS GIS Cut Line= 6
605305.336389571731426.972902432604700.206481308731241.732817352
 604619.56315878731078.835790589 603762.80296132730438.870273098
601760.703067303730892.898391157600848.399958491731155.871110424
#Sta/Elev= 30
8857.067184.60328950.975166.40629014.148141.30379077.321136.30789161.552139.2526
9716.606137.37349820.425132.85959884.903135.68299920.608131.12179946.108120.3412
9958.858118.781810048.11119.461710099.11114.957110126.69118.117510175.61134.4331
10191.17134.599910303.11126.195811225.13129.077211717.32123.028711823.39125.6955
12301.79125.642112363.31132.094912506.87127.986412547.88132.450612752.96137.4356
12783.72146.180512835.39149.148813210.04154.786713314.12161.496813758.08163.0195
#Mann= 3 , 0 , 0
8857.067  0.0532       08857.067  0.0532       013758.08  0.0532       0
#XS Ineff= 2 , 0
       09871.029        10205.46       0
Bank Sta=8857.067,13758.08
Exp/Cntr=0.3,0.1

Type RM Length L Ch R = 1 ,27681.99,986.874300,986.874300,986.874300
XS GIS Cut Line= 6
605054.930717736729949.160665914604417.963314086730047.265215382
604229.356283009730070.861585736603979.904945344730097.480129674
601578.588675112730692.579300061600705.581523716730975.795692682
#Sta/Elev= 30
9215.465282.2967 9286.32286.4453 9387.63246.83929438.226215.77989509.062200.3281
9701.303174.41699802.334151.21599832.643133.66159852.849130.89269883.107118.0154
    9999112.839410064.47132.306210154.99119.271310265.61111.398110357.47119.1945
10450.19117.254910584.13127.827310666.55 124.31611099.25127.3014 11727.7119.8012
12088.29123.840512191.32133.537512232.53124.991812294.34123.990612356.16126.0515
12397.37139.647513030.95155.931613188.64152.993313335.83157.396313692.66 155.965
#Mann= 3 , 0 , 0
9215.465    0.04       09215.465    0.04       013692.66    0.04       0
#XS Ineff= 2 , 0
       0                10100.66       0
Bank Sta=9215.465,13692.66
Exp/Cntr=0.3,0.1

Type RM Length L Ch R = 1 ,26695.11,530.290900,530.290900,530.290900
XS GIS Cut Line= 6
606061.500372414728423.987360186606057.081972718728452.075758249
605495.805141896728466.467471853603560.119661301729358.753715709
601825.918171227 730243.84410274 600417.24796792730649.370373425
#Sta/Elev= 30
 7871.52201.88518637.704157.33879113.556142.2402 9445.59136.50099738.335139.0331
9848.618129.20119925.816112.4658 9943.64114.40759991.074109.827810038.51111.4453
10091.24128.669510366.95128.201410477.23  143.2510510.31143.937810823.18136.0426
11193.68119.719711597.85116.979112293.94122.446612350.07106.184312394.98113.2805
12451.12128.708712603.29137.140812624.11143.371112728.17146.3645 12946.7 144.532
13227.66148.468513258.88145.901213539.84151.020213841.62146.127314005.78149.0868
#Mann= 3 , 0 , 0
 7871.52  0.0451       0 7871.52  0.0451       014005.78  0.0451       0
#XS Ineff= 2 , 0
       0                10275.64       0
Bank Sta=7871.52,14005.78
Exp/Cntr=0.3,0.1

Type RM Length L Ch R = 3 ,26508.62,,,
BEGIN DESCRIPTION:
END DESCRIPTION:
Bridge Culvert--1,0,-1,-1, 0
Deck Dist Width WeirC Skew NumUp NumDn MinLoCord MaxHiCord MaxSubmerge Is_Ogee
196.145450,138.000000,2.6,0, 60, 60, , , 0.95, 0, 0,0,,
 8464.13 8518.88 8679.10 9085.01 9362.73 9451.28 9555.75 9589.51 9847.26 9847.26
10215.2610215.2610248.9110261.1210316.1710382.2310547.3810635.4510767.7710834.11
10955.7111055.1411099.4311125.4911143.6511154.7111198.9311221.0411266.2111309.49
11360.0211364.7611375.8211383.4711406.9311408.9811420.0411431.0911464.2611486.37
11524.1911541.6511547.6411552.7011571.0911574.8111585.8711594.5511641.4511729.59
11740.6411983.8612063.6012193.9112448.1912724.9112820.2713032.1613253.8213737.53
  163.80  162.36  159.91  155.19  154.42  154.66  153.94  153.31  152.06  152.06
  150.28  150.28  150.12  149.49  148.79  148.76  147.25  147.32  145.47  145.64
  144.96  143.24  143.58  143.14  143.54  143.15  143.04  143.37  142.00  141.55
  142.84  142.01  133.09  127.75  118.42  117.84  116.82  116.46  116.85  117.63
  116.94  117.47  118.56  120.12  126.75  128.87  138.85  141.30  139.63  139.46
  139.83  137.85  137.98  137.10  136.94  134.90  133.79  133.15  134.65  141.92
 -836.20 -837.64 -840.09 -844.81 -845.58 -845.34 -846.06 -846.69 -847.94  144.56
  142.78 -849.72 -849.88 -850.51 -851.21 -851.24 -852.75 -852.68 -854.53 -854.36
 -855.04 -856.76 -856.42 -856.86 -856.46 -856.85 -856.96 -856.63 -858.00 -858.45
 -857.16 -857.99 -866.91 -872.25 -881.58 -882.16 -883.18 -883.54 -883.15 -882.37
 -883.06 -882.53 -881.44 -879.88 -873.25 -871.13 -861.15 -858.70 -860.37 -860.54
 -860.17 -862.15 -862.02 -862.90 -863.06 -865.10 -866.21 -866.85 -865.35 -858.08
 8464.13 8518.88 8679.10 9085.01 9362.73 9451.28 9555.75 9589.51 9827.67 9827.67
10195.6710195.6710248.9110261.1210316.1710382.2310547.3810635.4510767.7710834.11
10955.7111055.1411099.4311125.4911143.6511154.7111198.9311221.0411266.2111309.49
11360.0211364.7611375.8211383.4711406.9311408.9811420.0411431.0911464.2611486.37
11524.1911541.6511547.6411552.7011571.0911574.8111585.8711594.5511641.4511729.59
11740.6411983.8612063.6012193.9112448.1912724.9112820.2713032.1613253.8213737.53
  163.80  162.36  159.91  155.19  154.42  154.66  153.94  153.31  152.16  152.16
  150.38  150.38  150.12  149.49  148.79  148.76  147.25  147.32  145.47  145.64
  144.96  143.24  143.58  143.14  143.54  143.15  143.04  143.37  142.00  141.55
  142.84  142.01  133.09  127.75  118.42  117.84  116.82  116.46  116.85  117.63
  116.94  117.47  118.56  120.12  126.75  128.87  138.85  141.30  139.63  139.46
  139.83  137.85  137.98  137.10  136.94  134.90  133.79  133.15  134.65  141.92
 -836.20 -837.64 -840.09 -844.81 -845.58 -845.34 -846.06 -846.69 -847.84  144.66
  142.88 -849.62 -849.88 -850.51 -851.21 -851.24 -852.75 -852.68 -854.53 -854.36
 -855.04 -856.76 -856.42 -856.86 -856.46 -856.85 -856.96 -856.63 -858.00 -858.45
 -857.16 -857.99 -866.91 -872.25 -881.58 -882.16 -883.18 -883.54 -883.15 -882.37
 -883.06 -882.53 -881.44 -879.88 -873.25 -871.13 -861.15 -858.70 -860.37 -860.54
 -860.17 -862.15 -862.02 -862.90 -863.06 -865.10 -866.21 -866.85 -865.35 -858.08
Pier Skew, UpSta & Num, DnSta & Num=  ,9969.26, 2 ,9949.67, 2 , 0 , 0 , 0 ,,
    4.00    4.00
 -848.52  151.48
    4.00    4.00
 -848.43  151.57
Pier Skew, UpSta & Num, DnSta & Num=  ,10093.26, 2 ,10073.67, 2 , 0 , 0 , 0 ,,
    4.00    4.00
 -849.14  150.86
    4.00    4.00
 -849.04  150.96
BR Coef=-1 , 0 , 0 ,, 0 ,,,0.8,0,1,0,
WSPro=,,,, 1 ,,,, 0 ,,,, 0 ,,,,-1 ,-1 ,-1 , 0 , 0 , 0 , 0 , 0
BC Design=,, 0 ,, 0 ,,,,,,

Type RM Length L Ch R = 1 ,26164.82,650.418300,650.418300,650.418300
XS GIS Cut Line= 6
606055.720594404727745.909378246 603387.41909799728984.569161832
603027.626257777729171.661438778601214.270342857729984.793257773
 600343.57166937 730236.64824596600332.012747181730230.926007252
#Sta/Elev= 30
7399.742198.32138148.234182.48168456.618168.8077 8820.07178.39169183.523171.7727
 9821.96128.00659865.986114.71339899.006121.7996 9987.0697.0670710119.14101.3459
10324.71144.860710587.04134.201710643.39141.091110785.75131.818711030.01 133.264
 11194.499.3889911225.6798.7580811293.03114.478411470.08116.9776 11490.3109.4339
11567.02118.960611599.89114.118711610.85101.032811621.81 100.47811654.69114.6162
12114.98120.513612224.58134.956412421.85121.601612569.89142.742213659.76142.4583
#Mann= 3 , 0 , 0
7399.742  0.0662       07399.742  0.0662       013659.76  0.0662       0
#XS Ineff= 2 , 0
       0                10368.56       0
Bank Sta=7399.742,13659.76
Exp/Cntr=0.3,0.1

Type RM Length L Ch R = 1 , 25514.4,246.561700,246.561700,246.561700
XS GIS Cut Line= 6
603912.203706294727957.237718098603557.424749792728224.671949608
603359.846020909728352.919162795602163.627282787728963.513948253
601471.136124848729227.582789406600442.663798483729509.748596729
#Sta/Elev= 30
9191.859338.57429238.449325.64849413.769217.36719463.861191.09019564.044151.1865
9589.089 136.2939639.106118.29749671.546 112.3699819.596110.57079877.296116.0678
9933.546113.30259991.29799.2064710109.3898.3774610165.28 115.11110244.24116.2382
10312.39138.787610403.81 139.29810506.72130.1326 10655.1125.713510743.06112.9974
11195.32107.600211268.4993.6775911333.91110.425111355.56111.340912339.55110.7471
12484.78117.261212505.51125.581112557.33128.225612846.45124.2663 13023.7127.0455
#Mann= 3 , 0 , 0
9191.859  0.0474       09191.859  0.0474       0 13023.7  0.0474       0
#XS Ineff= 2 , 0
       0                10405.74       0
Bank Sta=9191.859,13023.7
Exp/Cntr=0.3,0.1

Type RM Length L Ch R = 1 ,25267.84,246.561600,246.561600,246.561600
XS GIS Cut Line= 6
 603780.33014825 727825.88727127603234.359678477728142.046756983
602023.039581358728704.801165745601490.853672534728921.371151596
600437.309241325729259.316986486599079.154374629729591.861243963
#Sta/Elev= 30
9271.923304.4382 9480.43 186.0549643.387124.24199700.632110.94319935.737  113.64
9990.738 99.028110100.43 94.567510166.23114.609310264.93111.598410330.76130.2932
10439.56133.923410485.91132.758810585.64115.952510740.79124.616611039.13122.2616
11302.25107.095811367.46 92.706911443.53105.554611530.21108.565212495.62107.8348
12558.35 117.57812662.86120.127212850.13120.746612860.53115.665312870.93121.2891
12943.66122.945713728.28125.050413974.75141.0757 14128.5136.7102   14319143.0016
#Mann= 3 , 0 , 0
9271.923  0.0517       09271.923  0.0517       0   14319  0.0517       0
#XS Ineff= 2 , 0
       0                10416.88       0
Bank Sta=9271.923,14319
Exp/Cntr=0.3,0.1

Type RM Length L Ch R = 1 ,25021.28,246.561700,246.561700,246.561700
XS GIS Cut Line= 6
603702.114854813727615.227414235603066.561441571727947.777720079
602005.772066385728425.769947693601193.387459815728759.861432537
600306.622917652729059.500458404598988.133452684729412.985146865
#Sta/Elev= 30
9258.449290.36849301.579279.50979485.593186.42159587.662 149.0899722.904127.9438
9789.894 125.6149878.477113.81639933.683114.9931 9988.8396.9306610098.5394.54486
10164.34114.907910197.24117.506310219.18109.193910295.95107.770310529.09120.2858
10899.19 125.12711052.74 124.19411140.47 108.85111412.74106.636111467.1990.99895
11543.17107.165711930.76111.231812101.63103.001912165.53107.872412420.04105.7314
12672.99117.589613517.92119.871213838.62135.723813910.96130.521414319.58138.5468
#Mann= 3 , 0 , 0
9258.449  0.0471       09258.449  0.0471       014319.58  0.0471       0
#XS Ineff= 2 , 0
       0                10423.94       0
Bank Sta=9258.449,14319.58
Exp/Cntr=0.3,0.1

Type RM Length L Ch R = 1 ,24774.72,246.561600,246.561600,246.561600
XS GIS Cut Line= 6
603619.968099028  727393.9788187602941.896806687  727733.6314338
601092.138342679 728538.94896315600466.271441907728771.829554334
599935.079411119728947.145053923598900.716502398729238.776829049
#Sta/Elev= 30
9242.427317.65789270.883314.78499508.471188.82329609.376145.56849721.099127.2221
9887.264110.53679931.396112.25539986.56197.2339110096.1594.1414710183.75115.3103
10205.65 114.38110227.55104.9354 10282.3104.813710358.95117.428310512.25119.3581
10599.85102.762110665.55120.3062 10917.4123.545711110.18115.244711223.36103.0404
11528.82105.001611639.2891.1333911734.75 104.92912475.42103.350212606.67108.1493
12666.14117.358513077.86113.685613538.48124.326513600.98118.386714320.64133.0739
#Mann= 3 , 0 , 0
9242.427  0.0484       09242.427  0.0484       014320.64  0.0484       0
#XS Ineff= 2 , 0
       0                 10418.3       0
Bank Sta=9242.427,14320.64
Exp/Cntr=0.3,0.1

Type RM Length L Ch R = 1 ,24528.15,246.561600,246.561600,246.561600
XS GIS Cut Line= 6
603536.474473357727169.102653518602668.178080559727588.404056907
601313.782232106728188.119059935600804.904308051728401.783769295
599844.994706959728756.795853987598813.994267851729068.099430546
#Sta/Elev= 30
9222.864309.95819460.334188.48119549.547155.03899671.637132.74719824.671119.4965
9870.757111.47739926.069 112.126 9981.3894.2634110091.7594.4511710154.97112.1935
10179.72114.2644 10223.5102.2823 10464.1112.653110540.66109.311410595.3499.70365
10825.01105.324611218.72101.441411413.75108.551911437.45104.670611711.57  103.11
11819.2789.4071311890.38 94.850311917.07103.588112510.41103.757812670.95112.1419
13243.98117.447213412.23117.693113454.29111.653813987.55125.996914321.09127.0558
#Mann= 3 , 0 , 0
9222.864  0.0507       09222.864  0.0507       014321.09  0.0507       0
#XS Ineff= 2 , 0
       0                10382.16       0
Bank Sta=9222.864,14321.09
Exp/Cntr=0.3,0.1

Type RM Length L Ch R = 1 ,24281.59,246.561700,246.561700,246.561700
XS GIS Cut Line= 6
603455.678325325726951.491694734602970.038905948727186.181571335
602251.318662554727492.018778235 600507.59349668728271.278176308
599765.565599084728558.803862154598733.615521193 728891.24443607
#Sta/Elev= 30
9211.744285.22289397.783202.84999558.221147.11669701.673126.71599833.003 119.748
9984.91281.8284710006.5281.6303110108.8283.3638310190.45106.493910277.41101.6321
10419.21109.595310736.5298.16451 10944.8104.979811219.6798.9834511604.48105.7087
11670.4498.2321111921.4895.3734411955.2388.1162211988.0990.6952712020.94101.3301
12628.64101.588512757.76105.198412832.88113.281213281.12112.712413348.14109.7754
13397.61100.675213556.42102.6166 13598.5111.815714060.24127.051114322.53121.1878
#Mann= 3 , 0 , 0
9211.744  0.0444       09211.744  0.0444       014322.53  0.0444       0
#XS Ineff= 2 , 0
       0                10352.83       0
Bank Sta=9211.744,14322.53
Exp/Cntr=0.3,0.1

Type RM Length L Ch R = 1 ,24035.03,246.561600,246.561600,246.561600
XS GIS Cut Line= 6
603366.400650471726711.037157059602942.014642477 726918.54171215
600812.514248401 727909.34880124600205.472000182728178.523752496
599409.813663661728488.398590192598662.036593169728733.842976525
#Sta/Elev= 30
9197.418236.89199299.619211.36349389.071173.24229588.909129.77549732.691118.0479
9827.70898.92093 9931.13 99.44239986.25281.8271910052.3181.2489910114.5386.46087
10162.05 100.57810304.71102.708410458.34113.816710667.13105.020111097.8397.40425
11562.74101.323811861.2195.5831211927.49 98.726311971.68 86.973812015.8790.40179
12037.87  101.1712769.72100.892412921.13112.997313349.93112.062413467.17106.3358
13636.96109.728813689.86106.853613732.18112.062414079.77122.743214323.77116.1045
#Mann= 3 , 0 , 0
9197.418  0.0486       09197.418  0.0486       014323.77  0.0486       0
#XS Ineff= 2 , 0
       0                10324.26       0
Bank Sta=9197.418,14323.77
Exp/Cntr=0.3,0.1

Type RM Length L Ch R = 1 ,23788.47,246.561600,246.561600,246.561600
XS GIS Cut Line= 6
603190.617348731726520.383525565601833.590668947727164.069063097
600542.898440003727803.601826176600128.625768036727994.832544431
599349.313858956728315.007859424598584.194688678728578.241874412
#Sta/Elev= 30
9276.853170.60319372.759167.3325 9506.45 150.4199695.172100.71899860.93295.38215
9927.132100.08089949.19997.579399971.26584.392139993.33280.6283310048.4385.04334
 10092.581.9735810169.63101.703410500.49100.983510533.71111.082910688.73103.6176
11133.9896.0405811559.0897.9308411827.5894.1011411971.5184.4911312027.8899.27579
12926.89101.074912952.74111.774613016.96 107.49813297.56106.250913394.13113.0021
13522.85106.5761 13639.9112.3033 13664.5106.092213870.82114.4911 14327.5111.7249
#Mann= 3 , 0 , 0
9276.853    0.04       09276.853    0.04       0 14327.5    0.04       0
#XS Ineff= 2 , 0
       0                10310.59       0
Bank Sta=9276.853,14327.5
Exp/Cntr=0.3,0.1

Type RM Length L Ch R = 1 ,23541.91,246.561600,246.561600,246.561600
XS GIS Cut Line= 6
603074.347341567726295.167606175601797.880529106726920.337265417
600801.478984535727446.978456825600059.929277927727817.460161492
599299.414492399728145.854582742598513.657298535728428.039625511
#Sta/Elev= 30
9286.772147.12139644.141118.09949734.76598.263199844.06692.824729921.81598.56524
9966.24383.115649987.52680.1271310099.3782.3048710132.6494.2780610165.91100.0967
10499.2799.4343810532.76109.421710577.41100.371811298.6794.7235311638.5897.07832
 11683.992.22312 11745.994.5715511876.2384.1925811921.2386.9130911966.2399.21265
11983.6799.4771112392.3196.6855113400.26103.764213583.06113.558613657.99 103.818
13797.14108.282514073.12109.204514104.94105.439114136.77110.387314327.74116.3362
#Mann= 3 , 0 , 0
9286.772  0.0454       09286.772  0.0454       014327.74  0.0454       0
#XS Ineff= 2 , 0
       0                10298.43       0
Bank Sta=9286.772,14327.74
Exp/Cntr=0.3,0.1

Type RM Length L Ch R = 1 ,23295.35,246.561700,246.561700,246.561700
XS GIS Cut Line= 6
602958.221382469726070.230709031601805.054947615726650.005064726
600563.627148181727349.960665375600000.920553058727642.794364363
599262.841190189727977.147676945598442.290060073728283.810357362
#Sta/Elev= 30
9294.582143.55319445.379129.62519703.661116.89149826.06893.569229870.51392.20158
9914.95797.836669970.51379.2511610092.7881.1134310107.8789.0718410153.6599.65879
 11458.195.1613111538.7890.3627611654.0292.9089111791.5182.0025711918.3199.25067
11959.3798.0532812031.78103.451212254.2296.4058112494.08 95.044813071.41103.2354
13503.49102.152613560.79111.314413603.87100.192413657.72106.873213946.78106.4855
14000.11102.790614021.44106.687414127.94107.907514212.47115.019214331.57115.5997
#Mann= 3 , 0 , 0
9294.582  0.0436       09294.582  0.0436       014331.57  0.0436       0
#XS Ineff= 2 , 0
       0                10284.16       0
Bank Sta=9294.582,14331.57
Exp/Cntr=0.3,0.1

Type RM Length L Ch R = 1 ,23048.79,246.561600,246.561600,246.561600
XS GIS Cut Line= 6
 602836.57150194725834.593932509601794.383299738726394.294136792
600653.358185053727091.553741693599959.343712002727477.167631209
599246.188044488727815.251688465598381.775512725728150.704210013
#Sta/Elev= 30
9300.901167.76749360.158154.00799520.607129.90369871.771103.17599916.79396.08353
9973.07178.1116410074.4580.3462210149.8798.92349 10423.4100.095710460.4496.27115
10997.6490.84873 11303.793.9487611597.3681.6567511667.45 87.446211725.8783.14522
11760.9191.0743111828.0789.3529411912.0496.4652411946.84103.728912165.74 102.211
12257.1994.0178512567.7993.4756413159.37102.172413579.3897.37778 13611.9102.9126
13741.6798.44187 13908.9109.7252 14158.8110.193514275.59118.7043 14332.1118.2521
#Mann= 3 , 0 , 0
9300.901  0.0421       09300.901  0.0421       0 14332.1  0.0421       0
#XS Ineff= 2 , 0
       0                10285.87       0
Bank Sta=9300.901,14332.1
Exp/Cntr=0.3,0.1

Type RM Length L Ch R = 1 ,22802.22,246.561600,246.561600,246.561600
XS GIS Cut Line= 6
602709.483396739725588.423272163601869.677742779726083.651748836
600729.255627722 726848.12701413600123.379751444727214.718428254
599247.140095711 727659.48344025598323.025149167728030.547734886
#Sta/Elev= 30
9298.448186.02129348.654173.11069409.813163.78679480.893 143.3819562.544129.1545
9730.711115.37419850.319110.46539922.67989.073149945.39578.241029979.46980.41249
10059.0777.9419510119.74101.876210139.3197.8924610197.6396.1633111013.7492.74765
11400.3880.83683 11556.387.0013411580.1690.9701311627.8990.9778311710.9684.72389
11752.68 91.805512637.92 92.930412977.5998.2400313064.24102.357613427.5199.15785
13471.1695.5555313634.84103.255313872.22104.557114086.55 115.29814333.97117.2668
#Mann= 3 , 0 , 0
9298.448  0.0427       09298.448  0.0427       014333.97  0.0427       0
#XS Ineff= 2 , 0
       0                10299.35       0
Bank Sta=9298.448,14333.97
Exp/Cntr=0.3,0.1

Type RM Length L Ch R = 1 ,22555.66,246.561700,246.561700,246.561700
XS GIS Cut Line= 6
602565.652872294725309.822413772600986.644126445726493.067045331
600252.711452603 726985.14101474599701.516347677727299.472057655
599236.775408864727531.054933891598261.044910669727931.277723297
#Sta/Elev= 30
  9268.4205.38739318.367200.20879416.696 174.7469634.835129.75059854.359110.0018
9921.94589.022539939.23979.6768610059.5777.9760910122.2597.2430710653.2194.31614
11019.6287.8235511218.9378.8114611329.7893.0801711378.9188.6323511610.8291.28261
11647.0686.2349811735.2791.5367411767.3488.1212111815.1291.7245212710.7492.25547
13070.4797.6276213173.7393.28304 13314.4100.121813653.51102.506413794.45111.7322
13902.69105.181214063.47113.720714224.25  110.8614256.11117.121814334.55 118.903
#Mann= 3 , 0 , 0
  9268.4  0.0452       0  9268.4  0.0452       014334.55  0.0452       0
#XS Ineff= 2 , 0
       0                10292.81       0
Bank Sta=9268.4,14334.55
Exp/Cntr=0.3,0.1

Type RM Length L Ch R = 1 , 22309.1,246.561600,246.561600,246.561600
XS GIS Cut Line= 6
 602371.06597805725049.227710888601191.300492376726137.570646033
 600329.86451748726782.350285485599420.028906137727309.909145936
598918.262767881727548.311369523598179.166222036727843.264081284
#Sta/Elev= 30
9248.875325.19639305.072281.55789352.201252.48619545.841163.04829680.307127.1211
9874.282103.85069956.53977.5246310060.13 78.505510125.2296.9135410473.2593.98216
10623.0587.86369 10914.988.9590710980.0586.1696511019.1378.2810311134.8186.03509
11695.5288.99309 11768.6 96.972311816.7587.4113712411.2993.8286812797.1990.24161
13000.2697.1829213443.64100.927913564.37109.484713651.31105.1512 13760.4110.0693
13900.72105.984214104.79112.218414243.85109.964114280.92122.199714335.04123.3241
#Mann= 3 , 0 , 0
9248.875  0.0567       09248.875  0.0567       014335.04  0.0567       0
#XS Ineff= 2 , 0
       0                10257.22       0
Bank Sta=9248.875,14335.04
Exp/Cntr=0.3,0.1

Type RM Length L Ch R = 1 ,22062.54,246.561600,246.561600,246.561600
XS GIS Cut Line= 6
602118.592658937724840.124041662601791.149186611725175.330823004
601258.072177798 725844.09100619600472.149375021726515.996477246
599295.860912919727233.099601343598067.638856441727760.123891443
#Sta/Elev= 30
9260.043 304.9559360.298238.69099428.049202.39769529.197183.12439622.037148.1654
9786.153110.58099834.34892.28992  9906.596.27441  9955.579.8073210003.73 77.0649
 10076.479.1196310138.4297.5778210259.0892.5703210290.7683.0964810330.0883.32017
10356.4492.3571510395.9887.7599410934.0187.4361910978.9776.2151511134.7285.19297
11542.3289.9308611788.8586.4824811827.0291.1989212541.2490.5638813230.49  98.699
13590.44111.1488 13662.7103.456314072.96112.893614233.76109.548614337.06123.7707
#Mann= 3 , 0 , 0
9260.043  0.0727       09260.043  0.0727       014337.06  0.0727       0
#XS Ineff= 2 , 0
       0                10244.34       0
Bank Sta=9260.043,14337.06
Exp/Cntr=0.3,0.1

Type RM Length L Ch R = 1 ,21815.98,246.561700,246.561700,246.561700
XS GIS Cut Line= 6
601918.945028335724674.771709591 601600.98154372725012.441563457
601026.746500731725761.464782119600277.159037113726418.309461996
599288.410214573727037.501884356597888.966644615727649.362714365
#Sta/Elev= 30
9234.905342.04159281.816335.78469393.971303.14439494.971231.98559650.281161.6703
9741.102 127.9239803.54686.639229853.39685.328879902.26594.781039962.11776.93386
10060.4575.6270410121.1696.6128810370.8184.72965 10975.886.8120811105.5474.27702
11145.4883.0575311315.2884.3779311367.0189.9839211721.77 85.604412105.8392.92085
12271.24 88.744413149.6496.1221113297.35106.646213480.51108.199113565.25107.0995
13611.7999.6531813914.72101.012814171.68118.347914214.37111.283114338.21113.7374
#Mann= 3 , 0 , 0
9234.905  0.0495       09234.905  0.0495       014338.21  0.0495       0
#XS Ineff= 2 , 0
       0                10229.69       0
Bank Sta=9234.905,14338.21
Exp/Cntr=0.3,0.1

Type RM Length L Ch R = 1 ,21569.42,246.561600,246.561600,246.561600
XS GIS Cut Line= 6
601757.709030151724541.232692674600666.324088275725745.242546558
599949.814837784726341.247314483599483.435083449726646.940201536
598852.047375441726991.942551717597669.207716227727484.482125491
#Sta/Elev= 30
9220.121279.8157 9346.64260.77139458.254277.8331 9499.62278.03589527.024268.8511
9581.833220.77869817.15484.241699832.48585.210639847.81595.354149924.392 94.5529
9940.32891.514569954.53969.36559 10020.466.6918110073.5467.5295510099.7885.95575
10151.52 93.422210345.5382.7256311014.1783.6943211139.8774.9622211254.1987.89767
11340.6582.0769211549.0989.6180211838.7487.6398312163.19 94.570512205.8990.00786
12393.4194.2995912907.5988.8482713905.93100.991714087.88109.607714339.01105.2526
#Mann= 3 , 0 , 0
9220.121  0.0478       09220.121  0.0478       014339.01  0.0478       0
#XS Ineff= 2 , 0
       0                10226.28       0
Bank Sta=9220.121,14339.01
Exp/Cntr=0.3,0.1

Type RM Length L Ch R = 1 ,21322.85,246.561600,246.561600,246.561600
XS GIS Cut Line= 6
601584.852209091724398.069067881601179.246904969724774.549517199
600514.313165605725548.445183218599725.452619702726197.556557983
598596.210304499726850.618076697597469.463127553 727306.26806365
#Sta/Elev= 30
9219.867209.86869246.153206.43179292.659210.23859552.906279.8148 9606.67285.4394
9621.566280.37399649.714234.81659677.405204.96589736.463152.46739826.72989.56161
9866.05979.494969930.133 85.25859980.52167.3383110003.33 66.146410102.4970.52525
10168.9686.7007710207.87  80.49110247.1484.5609110492.1579.48746   1093283.00105
11027.0172.5071211115.4183.71603 11444.887.5992612142.4887.0756112252.2393.30266
12672.2384.4763313058.0992.42706 13397.991.1047213865.3496.66289 14339.8107.6212
#Mann= 3 , 0 , 0
9219.867  0.0456       09219.867  0.0456       0 14339.8  0.0456       0
#XS Ineff= 2 , 0
       0                10220.37       0
Bank Sta=9219.867,14339.8
Exp/Cntr=0.3,0.1

Type RM Length L Ch R = 1 ,21076.29,246.561700,246.561700,246.561700
XS GIS Cut Line= 6
601457.539852411724292.626318485600957.978888869 724681.98740609
600016.285800248725580.479099095599340.729289234726075.004316419
598348.813325733726618.823965847597196.555436313727068.750833765
#Sta/Elev= 30
9196.285237.20829315.401179.48679364.777186.72419529.362232.07169615.084239.8136
9660.226213.4223 9665.85206.32979678.541  174.959692.706151.37739729.384113.6365
9768.47187.823239803.23477.98147  9892.685.213729934.92672.976379990.965 66.7206
10067.6768.4798910126.7386.6275110275.7775.1500810332.9785.1921610464.93 69.9532
10520.6769.0113410615.5671.9848610656.3983.2008710817.7485.1720212071.6287.71975
12118.8782.6779412671.3283.1539812840.2590.3454113499.2692.5233114340.13108.0443
#Mann= 3 , 0 , 0
9196.285  0.0453       09196.285  0.0453       014340.13  0.0453       0
#XS Ineff= 2 , 0
       0                10177.65       0
Bank Sta=9196.285,14340.13
Exp/Cntr=0.3,0.1

Type RM Length L Ch R = 1 ,20829.73,739.684800,739.684800,739.684800
XS GIS Cut Line= 6
601374.403082103724213.995964348600471.118997753724738.862166494
599531.205741763725467.382833079598858.218823254 725902.34782505
 598001.16955626726328.760077536 596833.86402601726752.197381839
#Sta/Elev= 30
9224.359224.75999295.363200.30659381.945158.58969416.578169.83189469.951179.1114
9563.519 193.4039598.964193.31389610.647186.45669645.368146.6884 9725.0181.24823
9878.89983.783069944.28767.3329110011.6666.1946510057.4967.5163810114.7885.90752
10196.3879.5848510243.5284.0509110267.0980.4635510352.2779.8479110655.4885.73725
10796.6880.0410910963.5683.0110311091.9278.17124 12010.382.9754612149.8979.05134
13062.9388.2272413139.6692.6114213263.0990.8527913313.8494.9402914462.97104.6826
#Mann= 3 , 0 , 0
9224.359  0.0492       09224.359  0.0492       014462.97  0.0492       0
#XS Ineff= 2 , 0
       0                10211.84       0
Bank Sta=9224.359,14462.97
Exp/Cntr=0.3,0.1

Type RM Length L Ch R = 1 ,20090.05,1232.808200,1232.808200,1232.808200
XS GIS Cut Line= 6
600922.503080159723444.813187405 600747.08383131723564.892240033
600572.342102528723734.356218502600203.681505084724240.218606234
599947.937482268724508.098163888596974.307546109725952.340329736
#Sta/Elev= 30
9143.368157.75379210.754156.55759246.844142.15199308.259137.49459417.955113.2061
9452.079109.99379566.451111.11139595.93597.772619642.81396.107399753.84782.53409
 9778.6886.080699807.37178.335599936.43674.419359985.69453.5733910094.7759.37132
 10158.575.1581510254.8180.2659410324.7375.37569 10722.374.5426211155.8780.58047
11433.7974.5917111511.6177.9643111825.6975.25253 12156.479.1781712178.6475.03288
12289.8174.8257412823.4279.4156612912.3686.2192512979.0682.6884613902.5593.75534
#Mann= 3 , 0 , 0
9143.368    0.04       09143.368    0.04       013902.55    0.04       0
#XS Ineff= 2 , 0
       0                10331.74       0
Bank Sta=9143.368,13902.55
Exp/Cntr=0.3,0.1

Type RM Length L Ch R = 1 ,18857.24,739.684900,739.684900,739.684900
XS GIS Cut Line= 6
601376.501596272723301.999354705600043.839831114723142.930288017
599632.113518178 723200.08073698 599335.72674036723244.682742968
598731.699745089723357.409140155598004.503398913723652.158808696
#Sta/Elev= 30
8125.584200.34368207.664204.35168278.161199.33468348.658172.39238399.013171.1643
 8469.51150.8246 8570.22 138.3868630.646118.13428892.49176.364678962.98880.96056
8993.20198.616719063.69899.724189194.621 110.726 9527.11112.58329555.493105.6718
9597.78174.297139617.973 67.95989880.465 72.95029941.14352.7365910001.8251.65501
10062.4953.3656310113.0572.2603910133.2873.2875710173.7368.8940110427.9969.98976
10550.0664.42306 10611.151.3757310692.4871.2543510912.6965.8558911582.2270.51949
#Mann= 3 , 0 , 0
8125.584  0.0426       08125.584  0.0426       011582.22  0.0426       0
#XS Ineff= 2 , 0
       09741.029        10218.79       0
Bank Sta=8125.584,11582.22
Exp/Cntr=0.3,0.1

Type RM Length L Ch R = 1 ,18117.55,986.246500,986.246500,986.246500
XS GIS Cut Line= 6
601373.832990289723033.112116963600788.973342955 723023.03465879
600399.907547027722947.376972526599384.401818395722331.827896923
598749.736146033722447.173919439598383.398091382722599.893755638
#Sta/Elev= 30
8160.859164.15358209.741155.57298229.746144.0504 8249.75146.19668269.754135.3389
8309.76298.988858369.77181.216088609.85982.153918629.89187.14654 8680.03 84.1145
8770.37967.700588820.72767.278459034.229110.38959343.452114.46679399.789108.6672
9434.22689.793099515.43867.346389670.65463.315199791.299 65.90929844.32560.28745
 9900.7842.2261710019.3942.9447110071.2259.7363610095.5559.3823510168.2546.54351
10192.15 52.181710216.0465.3423910466.0761.4715910577.8765.6094811376.51 65.0753
#Mann= 3 , 0 , 0
8160.859  0.0514       08160.859  0.0514       011376.51  0.0514       0
#XS Ineff= 2 , 0
       09625.798        10128.85       0
Bank Sta=8160.859,11376.51
Exp/Cntr=0.3,0.1

Type RM Length L Ch R = 1 ,17131.31,739.684900,739.684900,739.684900
XS GIS Cut Line= 6
601473.328053176722721.871151343601094.113469839722604.088177532
600830.688487679722432.248234823600320.685173094 721759.48348099
599489.965982139721754.983221188598539.092579601722121.013734272
#Sta/Elev= 30
8768.816111.30828920.932110.60228972.957124.71638983.362123.89848992.411118.4561
 9015.0788.818639025.70682.707829111.52677.931739140.027 64.77149164.85664.46484
9186.85369.221339315.07559.958279843.46858.630169879.51256.702159927.22939.72229
9942.91138.49389 9984.64 41.908710050.0340.2403710076.4550.2140810111.7257.97112
10386.5455.3923210516.5459.8217210616.5457.7373410766.5461.2426911046.5559.95258
11189.4663.3573411412.1559.0783711466.9362.5335311681.2460.8096312180.4764.46698
#Mann= 3 , 0 , 0
8768.816  0.0526       08768.816  0.0526       012180.47  0.0526       0
#XS Ineff= 2 , 0
       0 9796.17        10231.51       0
Bank Sta=8768.816,12180.47
Exp/Cntr=0.3,0.1

Type RM Length L Ch R = 1 ,16391.62,739.684900,739.684900,739.684900
XS GIS Cut Line= 6
602950.260120213722196.729674324601631.630037606721608.815936476
601199.892659098721447.429368585600542.337691486721384.563333735
599494.460566342721414.527802721598672.605253746721651.458191854
#Sta/Elev= 30
7765.285108.04147880.533106.2345 7913.38111.96857924.329106.75957946.226 109.733
7957.175104.84658064.21998.966338113.33488.35276 8236.1285.630358252.79679.38977
8263.74481.445098285.23576.287948384.18271.806448559.36571.102058581.26263.19916
8657.90559.644588734.54763.039898811.18956.285828931.627 54.30669483.013  53.389
  9845.359.314529925.50756.310379995.77534.8016810096.1738.0791310156.3555.72682
10588.3253.6735610938.4660.1226811268.5957.6641311378.6461.1688512234.5162.32683
#Mann= 3 , 0 , 0
7765.285   0.058       07765.285   0.058       012234.51   0.058       0
#XS Ineff= 2 , 0
       09768.056        10303.88       0
Bank Sta=7765.285,12234.51
Exp/Cntr=0.3,0.1

Type RM Length L Ch R = 1 ,15651.94,986.246600,986.246600,986.246600
XS GIS Cut Line= 6
602854.199764492721322.583009568601267.126596272720670.054910287
600920.816988885720696.957307473600416.433495522720678.759280488
 599530.43985036720853.250971928598439.487997472721182.811969444
#Sta/Elev= 30
7795.57461.416088282.88854.943578391.37356.685168489.00952.886529028.94153.04253
9115.15648.580179471.524 53.75179523.79149.72187 9914.9253.506729954.94737.38204
9974.97333.1569210075.1235.4654910095.1538.2701110135.1752.2987410155.1853.68299
 10185.249.1982910195.2154.4830310205.2155.3229710406.11 53.442110558.9957.40086
10650.7254.1395210691.4857.5116710895.3352.8811511241.8657.0784811491.9456.14433
11627.7560.0168211784.4458.7813311920.2463.0337112369.4458.5066312406.5362.06023
#Mann= 3 , 0 , 0
7795.574  0.0555       07795.574  0.0555       012406.53  0.0555       0
#XS Ineff= 2 , 0
       09692.043        10235.24       0
Bank Sta=7795.574,12406.53
Exp/Cntr=0.3,0.1

Type RM Length L Ch R = 1 ,14665.69,731.064400,731.064400,731.064400
XS GIS Cut Line= 6
604131.025486648 721431.20656389602143.732864916720110.404868573
 601036.36084637719710.037251517600450.478898138719716.784433126
599537.635707229  720004.1398689598111.192997098 720467.71322459
#Sta/Elev= 30
6250.51355.150537110.25841.365837218.323 44.13337309.56249.883687598.62144.46484
 7998.7948.874098176.73744.978228250.941 50.69848611.15652.875038699.14651.90303
8784.21446.784248975.61748.334049018.151 46.36259240.81149.56384 9347.7946.99591
9666.796 47.86379794.39850.999979955.62949.242719965.63223.30343 9995.6422.60802
10035.6423.2012510045.6449.0317110115.6551.7535710447.8546.8894210751.8853.29043
11060.3148.1521211633.3350.3014811685.9152.6500512295.7751.8442912857.0654.84153
#Mann= 3 , 0 , 0
6250.513  0.0598       06250.513  0.0598       012857.06  0.0598       0
#XS Ineff= 2 , 0
       09795.654        10145.93       0
Bank Sta=6250.513,12857.06
Exp/Cntr=0.3,0.1
